--- A111_00_00.prj (project) ---

Proj Title=A111-00-00
Current Plan=p01
Default Exp/Contr=.3,.1
English Units
Geom File=g01
Geom File=g02
Flow File=f01
Flow File=f02
Plan File=p01
Plan File=p02
Y Axis Title=Elevation
X Axis Title(PF)=Main Channel Distance
X Axis Title(XS)=Station
BEGIN DESCRIPTION:
Clear Creek Basin
Clear Creek Tributary 10.08
A111-00-00
Flood Hazard Model
10, 2, 1 & 0.2% Events
Filename: A111_00_00.prj
Prepared by: Perry Vaught	Date: 4-27-04
Reviewed by: __________	Date:
Status: (FINAL)
END DESCRIPTION:
DSS Export Rating Curves= 0
DSS Export Rating Curve Sorted= 0
DSS Export Volume Flow Curves= 0
DXF OffsetX= 0
DXF OffsetY= 0
DXF ScaleX= 1
DXF ScaleY= 10

--- A111_00_00.p01 (plan) ---

Plan Title=FEMA Effective June 2007
Version=Version 3.0.1  Mar 2001
Short Identifier=FEMAeff0607
Geom File=g01
Flow File=f01
Subcritical Flow
K Sum by GR= 0
Std Step Tol= 0.01
Critical Tol= 0.01
Num of Std Step Trials= 20
Max Error Tol= 0.3
Flow Tol Ratio= 0.001
Split Flow NTrial= 30
Split Flow Tol= 0.02
Split Flow Ratio= 0.02
Log Output Level= 0
Friction Slope Method= 0
Unsteady Friction Slope Method= 2
Secant Critical Depth
Global Vel Dist= 0 , 0 , 0
Global Log Level= 0
CheckData=True
Encroach Param=-1 ,0,0, 2
Computation Interval=1HOUR
Output Interval=1HOUR
Run HTab= 0
Run UNet= 0
Run PostProcess= 0
UNET Theta= 1
UNET ZTol= 0.02
UNET ZSATol= 0.1
UNET MxIter= 20
UNET MaxInSteps= 20
UNET DtIC= 0
UNET DtMin= 0
UNET MaxCRTS= 20
UNET WFStab= 2
UNET SFStab= 1
UNET WFX= 1
UNET SFX= 1
UNET Convert EG Bridges=-1
UNET Use Existing IB Tables=-1
Instantaneous Interval=1HOUR
Write IC File= 0
Write Velocity= 0
Write Detailed= 0

--- A111_00_00.p02 (plan) ---

Plan Title=Floodway
Version=Version 3.0.1  Mar 2001
Short Identifier=Floodway0607
Geom File=g02
Flow File=f02
Subcritical Flow
K Sum by GR= 0
Std Step Tol= 0.01
Critical Tol= 0.01
Num of Std Step Trials= 20
Max Error Tol= 0.3
Flow Tol Ratio= 0.001
Split Flow NTrial= 30
Split Flow Tol= 0.02
Split Flow Ratio= 0.02
Log Output Level= 0
Friction Slope Method= 0
Unsteady Friction Slope Method= 2
Secant Critical Depth
Global Vel Dist= 0 , 0 , 0
Global Log Level= 0
CheckData=True
Encroach Param=-1 ,0,0, 2
Encroach River=A111-00-00
Encroach Reach=A111-00-00_0020
Encroach Node=17126.63
       1 6775.05 6898.02
Encroach Node=16945.51
       1 4908.23 5050.48
Encroach Node=16120.32
       1 4953.27 5046.73
Encroach Node=14763.09
       1 4968.32 5068.03
Encroach Node=13475.86
       1 4925.31 5079.05
Encroach Node=12935.82
       1 4922.73 5030.24
Encroach Node=12913.91
       1 4922.73 5030.24
Encroach Node=12862
       1 4922.73 5030.24
Encroach Node=12822.08
       1 4922.73 5030.24
Encroach Node=12728.39
       1 4922.73 5080.69
Encroach Node=11598.32
       1  4933.8 5036.28
Encroach Node=10651.25
       1 4964.94 5036.68
Encroach Node=10007.5
       1 4933.02 5046.98
Encroach Node=9977.485
       1 4923.02 5036.98
Encroach Node=9916
       1 4923.02 5036.98
Encroach Node=9856.212
       1 4923.02 5036.98
Encroach Node=9807.355
       1 4933.21 5051.91
Encroach Node=9805
       1 4933.21 5051.91
Encroach Node=9639.737
       1 4933.21 5051.91
Encroach Node=9614
       1 4933.21 5051.91
Encroach Node=9589.726
       1 4933.21 5051.91
Encroach Node=9469.703
       1 4966.76 5033.24
Encroach Node=8386.021
       1 4966.33 5033.67
Encroach Node=7504.657
       1 4966.83 5033.17
Encroach Node=7416.087
       1  4969.2  5030.8
Encroach Node=7381.155
       1  4969.2  5030.8
Encroach Node=7379
       1  4969.2  5030.8
Encroach Node=7377.046
       1  4969.2  5030.8
Encroach Node=7308.124
       1  4969.2  5030.8
Encroach Node=7186.633
       1 4949.78 5028.41
Encroach Node=5857.266
       1 4961.06 5038.94
Encroach Node=4720.374
       1 4956.64 5029.16
Encroach Node=4690.362
       1    4956    5049
Encroach Node=4669
       1    4956    5049
Encroach Node=4650.352
       1    4956    5049
Encroach Node=4530.347
       1    4954    5087
Encroach Node=3840.003
       1 4859.19 5190.44
Encroach Node=3254.865
       1 4827.34 5101.35
Encroach Node=2739.518
       1 4969.42 5059.64
Encroach Node=2719.165
       1 4834.42 5059.64
Encroach Node=2706
       1 4969.42 5059.64
Encroach Node=2688.931
       1 4839.42 5059.64
Encroach Node=2608.866
       1 4930.84 5106.33
Encroach Node=2334.135
       1  4935.7 5082.04
Encroach Node=2312.034
       1  4935.7 5082.04
Encroach Node=2158
       1    4957    5039
Encroach Node=2044.285
       1    4850    5044
Encroach Node=1951.766
       1    4900    5044
Computation Interval=1HOUR
Output Interval=1HOUR
Run HTab= 0
Run UNet= 0
Run PostProcess= 0
UNET Theta= 1
UNET ZTol= 0.02
UNET ZSATol= 0.1
UNET MxIter= 20
UNET MaxInSteps= 20
UNET DtIC= 0
UNET DtMin= 0
UNET MaxCRTS= 20
UNET WFStab= 2
UNET SFStab= 1
UNET WFX= 1
UNET SFX= 1
UNET Convert EG Bridges=-1
UNET Use Existing IB Tables=-1
Instantaneous Interval=1HOUR
Write IC File= 0
IC Time=0
Write Velocity= 0
Write Detailed= 0

--- A111_00_00.f01 (steady flow) ---

Flow Title=FEMA Effective June 2007
Version=Version 3.0.1  Mar 2001
Number of Profiles= 4
Profile Names=10PCT_10yr, 2PCT_50yr, 1PCT_100yr, 0.2PCT_500yr
River Rch & RM=A111-00-00,A111-00-00_0020      ,17126.63
     339     522     619     906
River Rch & RM=A111-00-00,A111-00-00_0020      ,16945.51
     339     522     619     906
River Rch & RM=A111-00-00,A111-00-00_0020      ,16120.32
     410     632     749    1096
River Rch & RM=A111-00-00,A111-00-00_0020      ,14763.09
     492     757     897    1314
River Rch & RM=A111-00-00,A111-00-00_0020      ,13475.86
     531     817     968    1418
River Rch & RM=A111-00-00,A111-00-00_0020      ,12935.82
     539     830     984    1441
River Rch & RM=A111-00-00,A111-00-00_0020      ,12822.08
     640     986    1169    1711
River Rch & RM=A111-00-00,A111-00-00_0020      ,11598.32
     732    1127    1335    1955
River Rch & RM=A111-00-00,A111-00-00_0020      ,10651.25
     801    1234    1462    2140
River Rch & RM=A111-00-00,A111-00-00_0020      ,10007.5
     804    1239    1468    2149
River Rch & RM=A111-00-00,A111-00-00_0020      ,9977.485
     819    1262    1495    2189
River Rch & RM=A111-00-00,A111-00-00_0020      ,9469.703
     852    1312    1554    2276
River Rch & RM=A111-00-00,A111-00-00_0020      ,8386.021
     890    1370    1623    2377
River Rch & RM=A111-00-00,A111-00-00_0020      ,7186.633
     933    1437    1703    2494
River Rch & RM=A111-00-00,A111-00-00_0020      ,5857.266
     972    1498    1774    2598
River Rch & RM=A111-00-00,A111-00-00_0020      ,4720.374
    1004    1546    1831    2682
River Rch & RM=A111-00-00,A111-00-00_0020      ,3840.003
    1049    1616    1914    2803
River Rch & RM=A111-00-00,A111-00-00_0020      ,2608.866
    1074    1655    1960    2870
Boundary for River Rch & Prof#=A111-00-00,A111-00-00_0020      , 1
Up Type= 0
Dn Type= 3
Dn Slope=.002
Boundary for River Rch & Prof#=A111-00-00,A111-00-00_0020      , 2
Up Type= 0
Dn Type= 3
Dn Slope=.002
Boundary for River Rch & Prof#=A111-00-00,A111-00-00_0020      , 3
Up Type= 0
Dn Type= 3
Dn Slope=.002
Boundary for River Rch & Prof#=A111-00-00,A111-00-00_0020      , 4
Up Type= 0
Dn Type= 3
Dn Slope=.002
DSS Import GetInterval= 0
DSS Import GetPeak= 0
DSS Import FillOption= 0

--- A111_00_00.f02 (steady flow) ---

Flow Title=Floodway
Program Version=3.11
Number of Profiles= 2
Profile Names=1PCT_100yr, 1PCTFloodway_100yrFW
River Rch & RM=A111-00-00,A111-00-00_0020      ,17126.63
     619     619
River Rch & RM=A111-00-00,A111-00-00_0020      ,16945.51
     619     619
River Rch & RM=A111-00-00,A111-00-00_0020      ,16120.32
     749     749
River Rch & RM=A111-00-00,A111-00-00_0020      ,14763.09
     897     897
River Rch & RM=A111-00-00,A111-00-00_0020      ,13475.86
     968     968
River Rch & RM=A111-00-00,A111-00-00_0020      ,12935.82
     984     984
River Rch & RM=A111-00-00,A111-00-00_0020      ,12822.08
    1169    1169
River Rch & RM=A111-00-00,A111-00-00_0020      ,11598.32
    1335    1335
River Rch & RM=A111-00-00,A111-00-00_0020      ,10651.25
    1462    1462
River Rch & RM=A111-00-00,A111-00-00_0020      ,10007.5
    1468    1468
River Rch & RM=A111-00-00,A111-00-00_0020      ,9977.485
    1495    1495
River Rch & RM=A111-00-00,A111-00-00_0020      ,9469.703
    1554    1554
River Rch & RM=A111-00-00,A111-00-00_0020      ,8386.021
    1623    1623
River Rch & RM=A111-00-00,A111-00-00_0020      ,7186.633
    1703    1703
River Rch & RM=A111-00-00,A111-00-00_0020      ,5857.266
    1774    1774
River Rch & RM=A111-00-00,A111-00-00_0020      ,4720.374
    1831    1831
River Rch & RM=A111-00-00,A111-00-00_0020      ,3840.003
    1914    1914
River Rch & RM=A111-00-00,A111-00-00_0020      ,2608.866
    1960    1960
Boundary for River Rch & Prof#=A111-00-00,A111-00-00_0020      , 1
Up Type= 0
Dn Type= 3
Dn Slope=0.002
Boundary for River Rch & Prof#=A111-00-00,A111-00-00_0020      , 2
Up Type= 0
Dn Type= 3
Dn Slope=0.002
DSS Import GetInterval= 0
DSS Import GetPeak= 0
DSS Import FillOption= 0

--- A111_00_00.g01 (geometry) ---

Geom Title=A111-00-00 June 2007
Version=Version 3.0.1  Mar 2001

River Reach=A111-00-00,A111-00-00_0020
Reach XY= 30
     3189891.634    13767372.474     3190916.346    13766517.143
      3190942.25    13766188.999       3191041.5    13766083.999
        3191020.       13765930.      3190219.25       13765006.
      3190170.75    13764811.999       3190268.5       13764623.
        3191087.    13763908.999      3191187.75    13763003.999
        3191313.    13762771.999       3192586.5       13761678.
      3194950.75       13762168.      3195626.75    13762395.999
      3196809.75       13761891.       3196810.5       13761342.
        3197833.    13760187.999        3197795.    13759611.999
        3198063.    13759281.001       3198073.5    13758899.999
      3199013.75       13757826.      3199494.25       13758125.
      3199645.75    13757705.001       3199988.5       13757275.
        3200329.    13756427.999      3201383.75       13754671.
      3201866.25       13754327.      3203116.25       13754319.
        3203319.    13753232.001      3203478.25       13752949.

Type RM Length L Ch R = 1 ,17126.63,180.06,181.12,180.64
XS GIS Cut Line= 6
     3191880.331    13768474.686     3192623.995    13762315.207
     3192702.547    13761751.291      3192748.15    13761391.671
     3192728.709    13760794.547     3191764.314    13758546.583
#Sta/Elev= 30
       0   31.43  391.83   31.22  524.09   29.64  722.78   33.89  915.19   30.55
 1370.35   32.61 2281.53   28.68 2604.58   28.39 2782.92   27.31 3253.86   31.94
  3395.4   30.85 3891.65   31.38 4204.89   27.39 4501.21   29.95 4641.87   28.02
 4961.23   29.79 5161.73   27.12 5565.53   27.73 5681.38   30.05 5859.37   26.27
 5902.86   29.65 6009.17    30.1 6288.46   27.59 6597.73    31.2 6775.05   28.71
 6795.62   28.27 6840.92   15.48 6898.02   28.59 7461.05   30.2710179.62   27.62
#Mann= 9 ,-1 , 0
       0     .12       0  391.83     .07       0 2281.53     .15       0
 2604.58     .07       0  3395.4     .15       0 5565.53     .15       0
 6597.73     .07       0 6775.05    .035       0 6898.02     .12       0
Bank Sta=6775.05,6898.02
XS Rating Curve= 0
Exp/Cntr=.3,.1

Type RM Length L Ch R = 1 ,16945.51,830.65,825.19,823.43
XS GIS Cut Line= 6
     3192059.033    13768496.262       3192802.5    13762338.414
     3192881.135    13761773.903     3192928.535    13761400.556
     3192907.509     13760754.77     3191929.734    13758475.617
#Sta/Elev= 30
-1822.64   32.34-1308.89   31.43-1099.97   29.05 -842.22   33.76 -687.57   30.37
   26.87   30.15  129.63   30.33   519.7   29.96  783.84   27.31 1054.38   29.06
 1294.74   32.84 1729.87   29.41  1849.9   32.41 1988.96   30.84 2109.23   32.96
 2311.62   32.87 2516.13    26.9 2801.14   27.67  4136.9   28.95 4390.91   27.27
 4434.48   29.34 4733.66   31.21 4760.04   34.84 4782.83   33.54 4788.99   29.94
 4908.23   28.62 4949.52   28.17  5001.9   15.44 5050.48   29.22 8452.42   27.77
#Mann= 9 ,-1 , 0
-1822.64     .12       0-1308.89     .07       0   26.87     .15       0
  129.63     .07       0 1054.38     .15       0 2801.14     .15       0
  4136.9     .07       0 4908.23    .035       0 5050.48     .12       0
Bank Sta=4908.23,5050.48
XS Rating Curve= 0
Exp/Cntr=.3,.1

Type RM Length L Ch R = 1 ,16120.32,1333.76,1357.23,1318.28
XS GIS Cut Line= 6
      3193077.26    13768577.074     3193642.941    13762386.901
     3193686.248    13761940.943     3193749.902    13761427.783
     3193809.491    13760578.641     3192182.751    13758314.024
#Sta/Elev= 30
-1708.85   31.63 -386.96   29.83   95.03   31.08  337.44   28.75  435.99   29.25
  568.87   32.99  779.92   29.42 1061.08    31.4 1331.63   27.62 1702.25   32.89
 2151.98   32.62 2646.17   31.62 2783.77   29.18  2867.3   29.83 2970.05   26.86
 3810.63   26.11 3898.98   28.09 4242.55   25.62    4354   24.53 4428.82   19.05
  4716.1   20.82 4827.01   26.21 4953.27   25.35 4994.66   14.32 5046.73   26.25
 5146.72   27.84 6571.69   26.29 7898.24   27.31 8045.56   28.74 9111.88    26.5
#Mann= 5 ,-1 , 0
-1708.85     .07       0  779.92     .15       0 4242.55     .07       0
 4953.27    .035       0 5046.73     .12       0
#XS Ineff= 2 , 0
       0    4830    26.1               0
Permanent Ineff=
       F       F
Bank Sta=4953.27,5046.73
XS Rating Curve= 0
Exp/Cntr=.3,.1

Type RM Length L Ch R = 1 ,14763.09,1388.49,1287.23,1156.97
XS GIS Cut Line= 6
     3194750.178    13767573.971      3194963.29    13762476.986
     3194997.409    13762229.808     3195026.515     13762173.54
     3194820.302    13760786.797     3192519.242    13758106.952
#Sta/Elev= 30
 -381.57    29.8    -.15   29.82  529.61   29.03  593.24   23.05  823.86   22.69
  901.07   29.21 1018.97   30.02 2223.28   29.51 2343.04    26.8 2680.74   30.51
 2865.43   26.35 2930.92   28.53 2990.98   44.82 3007.65   46.67 3107.57   44.82
 3184.12   25.29 3447.63   24.27 3483.65   22.68 3561.47   25.35 3906.51   27.04
 4172.07   25.54  4231.8   23.67 4402.11   27.31 4700.57   21.32 4968.32   22.43
 5006.08    12.7 5031.68   19.63 5068.03    22.7 8788.31   28.32  9967.6   26.57
#Mann= 6 ,-1 , 0
 -381.57     .15       0    -.15     .07       0 3447.63     .15       0
 4172.07     .07       0 4968.32    .035       0 5068.03     .12       0
#XS Ineff= 2 , 0
       0    4815   22.96               0
Permanent Ineff=
       F       F
#Block Obstruct= 2 ,-1
  519.67  985.65   29.05    3420    3560    24.5
Bank Sta=4968.32,5068.03
XS Rating Curve= 0
Exp/Cntr=.3,.1

Type RM Length L Ch R = 1 ,13475.86,648.88,540.04,358.65
XS GIS Cut Line= 6
     3197158.776    13765327.513     3196427.303    13762931.762
     3196279.625    13762356.908     3196080.581    13761779.197
     3195216.583    13760737.055      3192690.68     13758000.74
#Sta/Elev= 30
 1674.04   28.48  2113.4   27.52 2464.89   25.49 2499.59   25.28 2537.77   14.95
 2566.05   11.24 2625.77   10.33 2707.18   11.03 2879.73   18.68 2928.69   25.71
 3881.87      24 4021.54   25.81 4165.21   21.71 4222.33   22.88 4318.02   25.04
 4573.82   20.89 4680.22   21.38 4758.08   15.81 4804.04   20.76 4925.31   22.07
 4963.68   20.13 5010.72   12.28 5036.32    20.7 5079.05   22.35 5804.03   24.23
 7233.44   26.46 9141.59   25.2410000.04   28.3310158.56   25.6510461.26   26.82
#Mann= 8 ,-1 , 0
 1674.04     .15       0  2113.4     .07       0 2464.89     .15       0
 4222.33     .07       0 4573.82     .12       0 4925.31    .035       0
 5079.05     .07       0 5804.03     .12       0
#Block Obstruct= 2 ,-1
 2482.81 2935.42   25.59    4120    4250      23
Bank Sta=4925.31,5079.05
XS Rating Curve= 0
Exp/Cntr=.3,.1

Type RM Length L Ch R = 1 ,12935.82,20.02,21.91,20.8
XS GIS Cut Line= 6
     3198643.683     13763633.66     3197111.399    13762292.022
     3196917.045    13762105.409     3196390.001    13761661.595
     3195920.999    13760874.529     3192897.795    13757865.908
#Sta/Elev= 30
 2420.24   23.28 2537.57   22.17 2933.52   24.19 2989.81   22.42 3074.38   24.29
 3341.42   22.89 3810.28   23.58 3934.75   25.04 3991.93   23.47 4449.07   24.13
 4546.19      21    4587   20.95 4683.76   24.36 4819.79   19.81 4922.73   19.56
 4986.79   16.33 4990.08   12.49 4999.75   11.25 5011.29   13.27 5013.21   15.98
 5030.24   19.25 5363.86   22.16 5609.16   23.28 6266.31   24.35 7414.57   22.92
 7812.89   24.19 7974.88    22.8 8209.33   24.1710141.91   25.1710596.97   26.87
#Mann= 8 ,-1 , 0
 2420.24     .07       0 3074.38     .12       0 3810.28     .15       0
 4546.19     .07       0 4922.73    .035       0 5030.24     .12       0
 5363.86     .07       0 5609.16     .12       0
#Block Obstruct= 1 ,-1
 4433.31 4673.57   24.06
Bank Sta=4922.73,5030.24
XS Rating Curve= 0
Exp/Cntr=.5,.3

Type RM Length L Ch R = 1 ,12913.91,80.06,91.83,93.7
XS GIS Cut Line= 6
     3198654.827     13763619.73     3197124.949    13762277.306
     3196930.377    13762090.483     3196405.437    13761648.429
     3195936.893    13760862.132      3192915.59    13757856.201
#Sta/Elev= 30
  2430.9   22.96 2563.23   22.01 2943.85   24.37 2993.54   22.03 3084.41    24.2
  3819.6   23.27 4455.57   23.62  4554.8   21.13 4595.54   20.91 4693.63   24.32
 4819.79   19.81 4922.73   19.56 4986.79   16.33 4989.77   13.23    4990   10.92
 4999.79   10.91 5010.95   10.91 5013.21   15.98 5030.24   19.25 5131.48   20.49
 5371.68   21.95 5535.06   22.08  5872.5   24.25 7376.46   22.88 7825.79   24.11
 7993.25   22.66 9965.69   26.4710125.44   24.9810444.98   27.4410599.75    26.9
#Mann= 9 ,-1 , 0
  2430.9     .07       0 3084.41     .12       0  3819.6     .15       0
  4554.8     .07       0 4922.73    .015       0 5030.24     .07       0
 5131.48     .12       0 5371.68     .07       0 5535.06     .12       0
#XS Ineff= 2 , 0
       0    4976   19.35    5023       0   19.35
Permanent Ineff=
       F       F
#Block Obstruct= 1 ,-1
 4450.72  4687.6   23.55
Bank Sta=4922.73,5030.24
XS Rating Curve= 0
Exp/Cntr=.5,.3

Type RM Length L Ch R = 2 ,12862   ,,,
BEGIN DESCRIPTION:
MEDICAL CENTER BLVD
END DESCRIPTION:
Bridge Culvert--1,0,-1,-1, 0
Deck Dist Width WeirC Skew NumUp NumDn MinLoCord MaxHiCord MaxSubmerge Is_Ogee
14,69,2.6,0, 11, 11, , , .95, 0, 0,0,,
    2358    2686    3110    3527    3819    4239    4719    4768    5077    5363
    5472
   22.81   23.16   23.71   22.75   23.54   23.41   24.21      20   20.56   22.23
   22.06
                                                                                
        
    2358    2686    3110    3527    3819    4239    4719    4768    5077    5363
    5472
   22.81   23.16   23.71   22.75   23.54   23.41   24.21      20   20.56   22.23
   22.06
                                                                                
        
Culvert=2,8,8.7,69,.012,.5,1,10,1,10.93,4995.15,10.89,4995.15,Culvert #1  , 0 ,14
Culvert Bottom n=.012
Culvert=2,8,8.95,69,.012,.5,1,10,1,10.93,5004.5,10.89,5004.5,Culvert #2  , 0 ,14
Culvert Bottom n=.012
BC Design=,, 0 ,, 0 ,,,,,,
BC HTab HWMax=27.44

Type RM Length L Ch R = 1 ,12822.08,80.06,93.7,97.96
XS GIS Cut Line= 6
     3198704.974    13763561.225      3197179.15    13762218.441
     3196983.703    13762030.779     3196467.181    13761595.765
      3196000.47    13760812.543     3192988.389    13757810.905
#Sta/Elev= 30
 2459.35   21.74 2866.51   23.83 2974.88   24.23 3013.31   21.54 3073.02   21.69
  3119.6   24.31 3656.05   22.09 4169.41   23.38 4576.56    21.3 4627.59   21.17
 4721.29    24.2 4819.79   19.81 4922.73   19.56 4986.79   16.33 4989.77   13.23
 4990.05   10.91 5010.82   10.91 5011.76   13.95 5013.21   15.98 5030.24   19.25
 5390.87    21.3 6057.86   24.11 7294.62   22.79 7866.01    23.8 8055.67   22.09
 9704.11   25.65 9983.46   25.3610027.14   24.1810398.87   27.6410602.47   26.94
#Mann= 7 ,-1 , 0
 2459.35     .15       0 2866.51     .07       0 4169.41     .15       0
 4576.56     .07       0 4922.73    .015       0 5030.24     .07       0
 5390.87     .12       0
#XS Ineff= 2 , 0
       0    4976   19.35    5023       0   19.35
Permanent Ineff=
       F       F
#Block Obstruct= 2 ,-1
  4448.2 4701.35   22.91    2990    3090    22.5
Bank Sta=4922.73,5030.24
XS Rating Curve= 0
Exp/Cntr=.5,.3

Type RM Length L Ch R = 1 ,12728.39,1009.4,1130.06,1010.24
XS GIS Cut Line= 6
     3198752.335    13763491.577     3197233.352    13762159.577
      3197037.03    13761971.075     3196528.926    13761543.101
     3196064.047    13760762.954     3193062.805    13757773.696
#Sta/Elev= 30
 2431.95      23 2579.97    26.1 2695.62   22.92 2918.02   23.18 2984.69   21.35
 3081.39   24.29 3499.03   24.33 3603.32   21.85 3675.25    23.5 4133.19   23.94
  4438.5   23.06 4538.24    20.6 4681.02   24.16  4783.2   19.74 4922.73   19.56
 4999.75   11.25 5011.18   13.28 5013.21   15.98 5080.69    19.8 5348.35    21.4
 5478.87   23.55 5598.32   22.12  6201.3    24.1 8046.64    21.9 9069.28   23.63
 9202.93   25.79 9293.54   24.11 9948.78   23.7510316.93   27.7110533.07   26.68
#Mann= 7 ,-1 , 0
 2431.95     .15       0 2918.02     .07       0 4133.19     .15       0
 4538.24     .07       0 4922.73    .035       0 5080.69     .07       0
 5348.35     .12       0
#Block Obstruct= 2 ,-1
 4363.63 4688.81   23.12    2940    3060    22.3
Bank Sta=4922.73,5080.69
XS Rating Curve= 0
Exp/Cntr=.3,.1

Type RM Length L Ch R = 1 ,11598.32,1089.25,947.07,768.04
XS GIS Cut Line= 6
     3199398.673    13762758.874     3197817.454    13761358.188
     3197293.444    13760876.956     3197008.346    13760647.673
     3195024.526    13759116.013     3193318.409    13757610.304
#Sta/Elev= 30
 2098.34   22.32 2496.92   22.92 2617.66   20.54 2736.07   22.78 3054.93   22.65
 3294.08   23.99 3884.69   22.47 4042.21    24.6 4169.06   22.91 4201.88   19.77
 4250.67   20.45 4358.91   23.72 4474.64   18.36 4619.55   20.28 4723.74   18.85
 4880.06   23.39  4933.8   20.93 4971.62    8.53 4995.73   17.45 5036.28   20.76
  5115.1   24.67 5326.34    26.1 5680.36   21.71 6154.28   23.76 6746.93   23.31
 6964.63   20.45  7359.6   21.58 8316.19   21.22 9990.23   24.8610069.95   25.05
#Mann= 11 ,-1 , 0
 2098.34     .12       0 2496.92     .07       0 2736.07     .12       0
 3054.93     .07       0 3294.08     .15       0 4250.67     .07       0
  4933.8    .035       0 5036.28     .07       0  7359.6     .15       0
 8316.19     .07       0 9990.23     .12       0
#XS Ineff= 1 ,-1
    4390    4800    21.9
Permanent Ineff=
       F
#Block Obstruct= 2 ,-1
 4024.16 4357.01   23.61    2530    2730      22
Bank Sta=4933.8,5036.28
XS Rating Curve= 0
Exp/Cntr=.3,.1

Type RM Length L Ch R = 1 ,10651.25,457.87,643.74,724.29
XS GIS Cut Line= 6
     3200287.389    13761742.005     3198225.188       13760204.
     3197974.497    13760121.877     3197733.642    13760144.624
     3197482.038    13760046.501     3193915.357    13757231.751
#Sta/Elev= 30
 2027.42   21.86 2116.69   20.35 2427.97   22.03 2554.15   19.68 2659.04   23.23
 3623.98   22.08 3841.69   19.33 3889.06   21.85 3932.26   19.97 3988.92   22.13
 4069.47      19 4303.26   22.22 4367.57    18.8 4462.02   18.04 4737.26   19.51
 4964.94   17.25 4987.49   11.29 4988.88     8.2 4990.63    7.71 5036.68    17.7
 5573.59   21.89 5638.38   19.43 7058.82    18.6 7451.83   20.64 8097.16   18.42
 8456.18   21.43    9520   21.03 9645.46   24.58 9790.68   22.38 9922.73   23.15
#Mann= 4 ,-1 , 0
 2027.42     .07       0 2659.04     .15       0 4964.94    .035       0
 5036.68     .07       0
#XS Ineff= 1 ,-1
    5600    8380      20
Permanent Ineff=
       F
#Block Obstruct= 2 ,-1
 3624.68 4302.49   22.04    2400    2610      22
Bank Sta=4964.94,5036.68
XS Rating Curve= 0
Exp/Cntr=.3,.1

Type RM Length L Ch R = 1 ,10007.5 ,39.04,30.02,32.51
XS GIS Cut Line= 6
     3200362.431    13761617.674     3199155.771    13760618.827
     3198424.356     13759970.26     3197422.233    13759109.336
     3197242.665     13758995.38     3194465.312    13756899.493
#Sta/Elev= 30
  1720.1   21.03 2168.01   19.06 2249.12   20.85 3168.05   22.58 3364.09    20.5
 3701.55   22.21    3780      25 3845.71   19.68 3945.43   22.35 4058.48   19.68
 4124.84   26.04 4403.11   20.05 4933.02   18.96 4951.79   16.05 4967.62    7.95
  4983.3       7 4998.53    7.88 5014.81   16.04 5046.98    19.6 5275.91   17.51
 5306.75   19.86 5505.83   20.26  5910.5   17.36 6673.13   20.69 6739.86   18.44
 7127.73   17.85  7289.9   21.71 7417.79   17.17 7527.25   19.95 9277.48   20.27
#Mann= 4 ,-1 , 0
  1720.1     .07       0 2249.12     .15       0 4933.02    .015       0
 5046.98     .07       0
#XS Ineff= 1 ,-1
    5520    9040    19.5
Permanent Ineff=
       F
#Block Obstruct= 1 ,-1
 2088.43    2352   21.29
Bank Sta=4933.02,5046.98
XS Rating Curve= 0
Exp/Cntr=.5,.3

Type RM Length L Ch R = 1 ,9977.485,139.43,121.27,121.99
XS GIS Cut Line= 6
     3200381.561    13761594.564     3199175.293    13760596.043
     3198443.911    13759947.504     3197440.012    13759085.088
     3197259.765    13758970.701     3194483.383    13756875.546
#Sta/Elev= 30
 1715.73   20.52 2111.54   22.39 2164.61   19.11 2244.84   20.27 2324.23   22.62
 3404.75   21.21 3778.85    33.8 3831.26   20.14 3938.24   22.34 4035.77   19.57
 4065.75   21.85 4088.22   31.08 4108.25   35.08 4150.83   35.06 4402.06   23.24
 4667.71   18.95 4923.02   18.96 4941.79   16.05 4957.79       7 4988.68       7
 5004.81   16.04 5036.98    19.6 5909.24    17.2 6671.87   20.94 6730.97   18.34
 7124.06    17.8 7288.64   21.45 7410.58   17.06 7511.36   19.91 9274.47   20.16
#Mann= 4 ,-1 , 0
 1715.73     .07       0 2244.84     .15       0 4923.02    .015       0
 5036.98     .07       0
#XS Ineff= 2 , 0
       0    4954    19.2    4992       0    19.2
Permanent Ineff=
       F       F
#Block Obstruct= 1 ,-1
 2064.91    2352   21.86
Bank Sta=4923.02,5036.98
XS Rating Curve= 0
Exp/Cntr=.5,.3

Type RM Length L Ch R = 2 ,9916    ,,,
BEGIN DESCRIPTION:
528
END DESCRIPTION:
Bridge Culvert--1,0,-1,-1, 0
Deck Dist Width WeirC Skew NumUp NumDn MinLoCord MaxHiCord MaxSubmerge Is_Ogee
1,120,2.6,0, 23, 23, , , .95, 0, 0,0,,
    1664    2074    2518    2974    3296    3760    4026    4100    4424    4771
    4893    4922 4945.06 5015.39 5041.63 5080.99 5120.68    5173    5298    5607
    5912    6680    8250
   20.68   22.52   21.68   21.73   23.19   38.92   39.27   36.81   26.04   20.36
   19.96   19.93   20.47   20.18   19.95   19.68   19.44   19.32   19.84   19.03
   19.03      21      19
                                              33      33      33
                                                                                
                        
    1664    2074    2518    2974    3296    3760    4026    4100    4424    4771
    4893    4922 4945.06 5015.39 5041.63 5080.99 5120.68    5173    5298    5607
    5912    6680    8250
   20.68   22.52   21.68   21.73   23.19   38.92   39.27   36.81   26.04   20.36
   19.96   19.93   20.47   20.18   19.95   19.68   19.44   19.32   19.84   19.03
   19.03      21      19
                                              33      33      33
                                                                                
                        
Multiple Barrel Culv=2,8,8,120,.012,.5,1,10,1,7.07,6.96, 3,Culvert #1  , 0 ,1
    4964    4964    4973    4973    4982    4982
Culvert Bottom n=.012
BC Design=,, 0 ,, 0 ,,,,,,
BC HTab HWMax=35.08

Type RM Length L Ch R = 1 ,9856.212,44.85,48.86,30.1
XS GIS Cut Line= 6
     3200441.929     13761534.66     3198645.855    13759959.745
     3198437.012    13759761.409      3198210.43    13759595.576
     3197433.482    13758919.192      3194641.92    13756781.134
#Sta/Elev= 30
 1713.21   20.69 2095.93    22.5  2234.4   19.02 2275.21   22.33 2313.54   22.06
 3050.48   20.22 3330.59   22.68 3535.76   20.76 3773.28   27.97 3829.52   20.22
 3943.36   22.15 4040.86    19.8  4070.9   21.61 4109.89   28.52 4308.93   19.24
 4570.54   21.61 4923.02   18.96 4941.79   16.05 4957.79       7 4988.68       7
 5004.81   16.04 5036.98    19.6 6473.65   19.49 6707.67   16.87 6818.36   18.12
 6866.01   15.79 7326.09   19.01 7393.96   16.89 7568.84   18.88 9217.32   19.81
#Mann= 4 ,-1 , 0
 1713.21     .07       0 2313.54     .15       0 4923.02    .015       0
 5036.98     .07       0
#XS Ineff= 2 , 0
       0    4954   19.28    4992       0   19.28
Permanent Ineff=
       F       F
Bank Sta=4923.02,5036.98
XS Rating Curve= 0
Exp/Cntr=.5,.3

Type RM Length L Ch R = 1 ,9807.355,377.08,167.62,50.91
XS GIS Cut Line= 6
     3200445.225      13761530.9     3198649.226    13759956.051
     3198195.663    13759525.307     3197977.043    13759327.473
     3197710.383     13759130.15     3194644.961    13756777.165
#Sta/Elev= 30
 1723.99   20.78 2104.67   22.49 2237.11   19.04 2324.41   22.15 3060.93   20.03
 3335.97   22.63  3570.3   20.55 3783.73    26.5 3845.48   19.98 3954.36   22.15
  4053.4   19.74    4122   26.96 4304.56   18.73 4521.83   18.13  4601.2   21.25
 4691.01    18.4 4717.74   20.58 4783.74   17.13 4965.43   18.41 4982.21     8.3
 4999.63    5.43 5017.98    7.47 5034.57   18.43 6523.23   19.43 6726.92   16.92
 6833.04   18.16 6877.22   15.47  7337.3   18.73 7404.42   16.89 9229.19   19.81
#Mann= 4 ,-1 , 0
 1723.99     .07       0 2324.41     .15       0 4965.43    .015       0
 5034.57     .07       0
#Block Obstruct= 3 ,-1
    4260    4590    19.1    6000    8640    18.7    4650    4700    18.7
Bank Sta=4965.43,5034.57
XS Rating Curve= 0
Exp/Cntr=.5,.3

Type RM Length L Ch R = 5 ,9805    ,,,
BEGIN DESCRIPTION:
Downstream of 528
END DESCRIPTION:
IW Pilot Flow=0
#Inline Weir SE= 17
4965.985   18.39 4977.14   18.414988.906    18.44989.169   14.924994.415   14.94
4994.606   10.814994.866   10.18 4997.84   10.174997.934    7.535000.396    7.46
 5003.88    7.515004.121   10.175007.136   10.175007.325   14.955012.896   14.96
5013.015   18.43 5034.57   18.43
IW Dist,WD,Coef,Skew,MaxSub,Min_El,Is_Ogee,SpillHt,DesHd
2,.1,3.3,0,.95,, 0 ,,,0,0,

Type RM Length L Ch R = 1 ,9639.737,70.65,50.01,53.46
XS GIS Cut Line= 6
     3200688.154    13760874.154      3198657.58    13759191.081
     3198269.138     13759196.98     3198105.556    13759203.059
     3197890.521    13759218.411     3194824.352    13756672.322
#Sta/Elev= 30
 1773.98   21.15 1926.62   21.64 1964.56   18.53 1989.73   22.92 2042.33   19.66
 2365.23   22.11 2467.15   20.33    2695   22.09 2784.36   18.72 2889.52   22.43
 2980.29   20.82 3522.35   21.38 3618.96   17.94 3757.45   21.43 3853.33   17.83
 4142.99   16.34 4933.21   19.64 4966.76    17.8 4984.05    7.26 4997.59    5.59
 5016.71    7.28 5033.24   17.67 5051.91   19.74 6111.13   20.16 6777.98   17.45
  6964.6   19.71    8099   19.69 8654.27   17.43 8958.67   20.69 9164.63   19.45
#Mann= 4 ,-1 , 0
 1773.98     .07       0 2365.23     .15       0 4933.21    .015       0
 5051.91     .07       0
#XS Ineff= 2 , 0
       0    4967    18.4    5033       0    18.4
Permanent Ineff=
       F       F
#Block Obstruct= 1 ,-1
    3975    4350    17.4
Bank Sta=4933.21,5051.91
XS Rating Curve= 0
Exp/Cntr=.5,.3

Type RM Length L Ch R = 3 ,9614    ,,,
BEGIN DESCRIPTION:
ACCESS RD
END DESCRIPTION:
Bridge Culvert--1,0,-1,-1, 0
Deck Dist Width WeirC Skew NumUp NumDn MinLoCord MaxHiCord MaxSubmerge Is_Ogee
1,48,2.6,0, 19, 19, , , .95, 0, 0,0,,
    3614    3735    3907    4140    4413    4675    4853 4892.33    4933 4967.68
 4967.82 4999.56 5031.35 5031.36 5051.41 5082.98 5119.52    5159    5228
   18.06   21.24   18.34   16.62   18.66   18.36   18.19   18.33   19.71   20.14
   20.17   20.24   20.14   20.17   20.13   20.03   19.93   19.79   19.41
                                                                           17.18
   17.18   17.18   17.18   17.18
    3614    3735    3907    4140    4413    4675    4853 4892.33    4933 4967.68
 4967.82 4999.56 5031.35 5031.36 5051.41 5082.98 5119.52    5159    5228
   18.06   21.24   18.34   16.62   18.66   18.36   18.19   18.33   19.71   20.14
   20.17   20.24   20.14   20.17   20.13   20.03   19.93   19.79   19.41
                                                                           17.18
   17.18   17.18   17.18   17.18
BR Coef=-1 , 1 , 0 ,1.25, 0 ,,,.8,-1,2,6,
WSPro=,,,, 1 ,,,, 0 ,,,, 0 ,,,,-1 ,-1 ,-1 , 0 , 0 , 0 , 0 , 0
BC Design=,, 0 ,, 0 ,,,,,,
BC HTab HWMax=22.92

Type RM Length L Ch R = 1 ,9589.726,141.03,120.02,128.4
XS GIS Cut Line= 6
     3200720.062    13760835.659      3198655.97    13759123.876
     3198268.509     13759139.83     3198103.041    13759153.118
     3197906.926    13759167.042     3194856.294    13756633.855
#Sta/Elev= 30
 1734.13   20.95 1891.67   21.27 1923.22   18.48 1955.13   22.79 2002.61   19.62
 2338.91    22.8 2402.59   20.32 2547.82    21.5 3459.31    20.4 3570.68    17.6
 3704.54   21.22 3808.75   17.78 3959.39   18.87 4105.22   16.33 4443.28   18.89
 4933.21   19.64 4966.76    17.8 4984.05    7.26 4997.59    5.59 5016.71    7.28
 5033.24   17.67 5051.91   19.74 5900.72   18.87 5974.17    20.2 6752.38   17.43
 6922.91   19.58 8479.92   19.85 8768.98   17.56 8977.25   20.81 9131.35   19.37
#Mann= 4 ,-1 , 0
 1734.13     .07       0 2547.82     .15       0 4933.21    .015       0
 5051.91     .07       0
#XS Ineff= 2 , 0
       0    4967   19.11    5033       0   19.11
Permanent Ineff=
       F       F
#Block Obstruct= 1 ,-1
    3990    4280    17.4
Bank Sta=4933.21,5051.91
XS Rating Curve= 0
Exp/Cntr=.5,.3

Type RM Length L Ch R = 1 ,9469.703,776.07,1083.68,1141.59
XS GIS Cut Line= 6
      3200796.64     13760743.27     3198690.158    13759003.079
     3198307.255    13759016.754     3198097.006    13759033.259
     3197946.298    13759043.758     3194973.363    13756573.329
#Sta/Elev= 30
 1636.99   20.99 1794.16   20.96 1819.71   17.97 1845.21   21.94 1890.16   19.57
 2010.59   22.36 2250.64   21.88 2307.58   19.77 2537.52   21.84 2738.42   19.55
 3479.42    17.6 3615.51    21.1 3710.86   17.29 3889.16   18.93 4012.82    16.3
 4460.03   19.65 4789.57   19.69 4819.74   16.45 4955.25   19.89 4966.76    17.8
 4984.05    7.26 4997.59    5.59 5016.71    7.28 5033.24   17.67  5854.2   20.06
 6735.87   17.18 6838.09   19.21 7482.01   19.89 8901.35   17.68 8979.83   19.06
#Mann= 4 ,-1 , 0
 1636.99     .07       0 2738.42     .15       0 4966.76    .015       0
 5033.24     .07       0
#Block Obstruct= 2 ,-1
    3912    4185    17.7    4800    4865    17.7
Bank Sta=4966.76,5033.24
XS Rating Curve= 0
Exp/Cntr=.3,.1

Type RM Length L Ch R = 1 ,8386.021,191.78,881.36,731.88
XS GIS Cut Line= 6
     3201411.915    13760445.259     3198794.184    13758273.637
     3198725.747    13758216.883     3198674.989     13758172.64
     3198602.869    13758113.346      3195908.42    13755984.469
#Sta/Elev= 30
  1475.3   19.45 1796.15   19.69  1904.6   18.13 1940.07   20.51 1954.61   20.41
 1990.27   17.87 2007.99    18.7 2111.51   19.04 2750.57   17.86 3143.34   18.68
 3438.11   17.83 3487.99   18.42 3620.73   16.62 3672.65   19.26 3726.66   19.28
 3763.97   18.89 3847.09   15.98 4602.48   19.06 4966.33   17.51 4985.99    5.17
 5002.35    4.68 5015.28    5.11 5033.67   17.45 5052.97   16.98  5064.8   18.12
 5413.09   18.41 5641.35   17.07  6445.1   17.91 7371.85   16.93 8560.12   18.53
#Mann= 4 ,-1 , 0
  1475.3     .07       0 2750.57     .15       0 4966.33    .015       0
 5033.67     .07       0
#Block Obstruct= 1 ,-1
    3560    4230    17.3
Bank Sta=4966.33,5033.67
XS Rating Curve= 0
Exp/Cntr=.3,.1

Type RM Length L Ch R = 1 ,7504.657,96.35,88.57,85.14
XS GIS Cut Line= 6
     3201458.825    13760271.021     3199120.006    13758314.186
     3199334.227    13758034.451     3199357.369    13758002.142
     3199187.021    13757771.366     3196968.828    13755425.845
#Sta/Elev= 30
 1632.96   26.55 1683.84   24.57 1732.68   19.17 1883.61   20.03 1985.23   18.39
 2024.95   20.72 2067.54   17.73 2109.11   20.02 2302.41   19.23 2429.18   20.46
 2483.59   18.56 2594.06   18.08 2876.82   19.35 2944.26    18.2 3309.63      17
 3564.16   17.74 3670.64   16.34 3767.64   19.86 3928.67   16.45  3977.8   17.42
 4129.64   16.35 4444.03   17.29 4680.37   19.05 4868.24   19.03 4966.83   16.61
 4981.18    7.49 5001.19    4.21 5021.83    7.55 5033.17   16.94 8589.66   17.15
#Mann= 4 ,-1 , 0
 1632.96     .07       0 3928.67     .15       0 4966.83    .015       0
 5033.17     .07       0
#Block Obstruct= 5 ,-1
 3069.13 3774.73   17.77    3880    4324   17.25    5140    5265      17
    5370    5960    16.8    7031    8000    16.8
Bank Sta=4966.83,5033.17
XS Rating Curve= 0
Exp/Cntr=.3,.1

Type RM Length L Ch R = 1 ,7416.087,57.1,34.93,24.74
XS GIS Cut Line= 6
     3201512.486    13760076.895     3199323.597    13758287.948
     3199411.159    13758067.716     3199395.239    13758004.035
     3199273.182    13757765.229     3197365.376    13755213.268
#Sta/Elev= 30
 1989.89   19.94 2133.17    19.8 2250.38   17.91 2282.34   20.44 2332.61   17.82
 2395.47   19.43 2722.18    19.7 2785.47   17.78  3147.6   19.75 3198.58   17.81
  3313.6   17.13 3430.72   18.35 3507.84   17.03 3800.62   17.51 3951.83   15.98
 4002.45   16.43 4035.78   19.58 4056.01   19.84 4143.92   18.53 4197.55   15.49
 4228.87   16.28  4816.9   17.98 4870.76   17.93  4969.2   15.65 4995.08    3.94
 5002.86    3.94 5009.73    7.99  5030.8   15.81 5191.67   17.08 8575.12   16.95
#Mann= 4 ,-1 , 0
 1989.89     .07       0 4228.87     .15       0  4969.2    .015       0
  5030.8     .07       0
#Block Obstruct= 3 ,-1
 3818.83 4135.88   17.63    4156    4590    16.9    5920    7919   16.55
Bank Sta=4969.2,5030.8
XS Rating Curve= 0
Exp/Cntr=.5,.3

Type RM Length L Ch R = 1 ,7381.155,4.47,4.11,4.36
XS GIS Cut Line= 6
     3201579.452    13760076.677     3199370.135    13758283.009
     3199425.783    13758108.111     3199413.549    13758004.378
     3199287.543    13757751.261     3197391.022    13755171.188
#Sta/Elev= 30
 2001.77   19.98 2192.62   19.73 2309.92   17.88 2341.91   20.42 2395.83   17.84
 2453.66   19.32 2789.33   19.54 2868.13    17.6 3211.14   19.59 3256.21   17.93
 3386.12   17.05 3501.56   18.31 3562.89    17.1 3907.06   17.43 4018.04   15.91
  4070.5   16.48 4109.81   19.83 4210.26   18.51  4252.1   16.11 4262.32   15.52
 4626.62   17.36 4892.41   17.26  4969.2   15.65 4995.08    3.94 5002.86    3.94
 5009.73    7.99  5030.8   15.81 5215.41   17.08 7344.27   16.39 8620.39   17.02
#Mann= 4 ,-1 , 0
 2001.77     .07       0  4252.1     .15       0  4969.2    .015       0
  5030.8     .07       0
#XS Ineff= 2 , 0
       0 4982.93   15.81 5015.82       0   15.81
Permanent Ineff=
       F       F
#Block Obstruct= 3 ,-1
 3818.83 4135.88   17.63    4230    4590    16.9    5920    7919   16.55
Bank Sta=4969.2,5030.8
XS Rating Curve= 0
Exp/Cntr=.5,.3

Type RM Length L Ch R = 5 ,7379    ,,,
IW Pilot Flow=0
#Inline Weir SE= 14
4966.678   15.824982.919   15.814982.977   13.544991.778   13.554991.958   12.49
4994.889   12.474994.889    7.455003.922    7.455003.922   12.485007.199   12.45
5007.254   13.565015.821   13.575015.822    15.8    5031   15.83
IW Dist,WD,Coef,Skew,MaxSub,Min_El,Is_Ogee,SpillHt,DesHd
2,.1,4.55,0,.95,, 0 ,,,3,3,

Type RM Length L Ch R = 1 ,7377.046,99.49,68.922,56.93
XS GIS Cut Line= 6
     3201581.973    13760073.572     3199374.761    13758281.612
     3199429.859    13758108.523      3199417.44    13758003.219
      3199290.97     13757749.17     3197394.245    13755168.819
#Sta/Elev= 30
 2005.82   19.98 2196.25   19.72 2313.55   17.88 2345.54   20.42 2399.83   17.84
 2457.14   19.31 2794.24   19.53 2874.28   17.58 3209.43   19.57 3259.52   17.95
 3391.28   17.04  3495.9   18.23  3565.8    17.1 3829.08   17.66 4022.47    15.9
 4075.43    16.5 4112.05   19.83 4214.68    18.5 4255.59   16.15 4266.52   15.52
 4629.88   17.36 4894.89   17.29  4969.2   15.65 4993.93    4.54 5002.86    3.94
 5009.73    7.99  5030.8   15.81 5217.24   17.08 7341.38   16.39  8622.8   17.04
#Mann= 4 ,-1 , 0
 2005.82     .07       0 4255.59     .15       0  4969.2    .015       0
  5030.8     .07       0
#XS Ineff= 2 , 0
       0 4982.93   15.81 5015.82       0   15.81
Permanent Ineff=
       F       F
#Block Obstruct= 3 ,-1
 3818.83 4144.22   17.57    4210    4600    16.6    5920    7920    16.6
Bank Sta=4969.2,5030.8
XS Rating Curve= 0
Exp/Cntr=.5,.3

Type RM Length L Ch R = 1 ,7308.124,258.83,121.49,104.69
XS GIS Cut Line= 6
      3201662.73    13759967.181     3199642.181     13758360.31
     3199512.731    13758194.276     3199421.803    13757930.039
     3199324.184    13757698.988     3197490.424    13755153.258
#Sta/Elev= 30
 2126.85   18.62 2395.33   19.25 2415.48   18.22 2458.87   19.78 2504.67   17.58
 2555.56   18.95 2958.07   19.16 3070.32   17.37 3236.32   18.91 3518.27   17.32
 3802.22   18.21 3912.45   17.19 4074.82   17.48 4152.79   15.34 4195.82   15.84
 4233.39   19.08 4257.56   19.57 4330.22   18.89 4387.79   16.07 4566.81   18.08
 4775.38   16.89 4906.17   17.19  4969.2   15.65 4993.93    4.54 5002.86    3.94
 5009.73    7.99  5030.8   15.81 5216.53   17.08 7842.95   16.39 8586.69   17.42
#Mann= 5 ,-1 , 0
 2126.85     .07       0 4387.79     .15       0 4775.38     .07       0
  4969.2    .015       0  5030.8     .07       0
#Block Obstruct= 3 ,-1
 3818.83    4270   17.57    4333    4600    16.6    5920    8100    16.6
Bank Sta=4969.2,5030.8
XS Rating Curve= 0
Exp/Cntr=.5,.3

Type RM Length L Ch R = 1 ,7186.633,1312.65,1329.37,989.41
XS GIS Cut Line= 6
     3202128.974    13759064.753     3199610.703    13758037.826
      3199541.58    13758019.289     3199472.166    13757994.199
     3199423.946    13757690.335     3197679.186    13755057.263
#Sta/Elev= 30
 2195.21   18.58 2311.09   17.03 2829.94   20.24 3064.16   18.23 3398.17   18.08
 3479.87    16.9 4157.93   16.72 4217.61   16.45 4252.53    19.5 4369.57   18.12
 4396.51   15.56 4440.04   16.79 4778.11   17.56 4949.78   15.46 4975.77   14.66
 4992.86    6.88 4993.24    5.75 4999.15    3.64    5006     3.6 5006.23    6.62
 5013.01    7.55 5028.41   15.48 5164.11   17.07  8345.5   17.15 8404.08   15.13
 8422.07   10.03 8440.06    7.56 8458.06    7.88 8499.43   16.67 8526.57   16.83
#Mann= 5 ,-1 , 0
 2195.21     .07       0 3398.17     .12       0 4157.93     .07       0
 4949.78    .015       0 5028.41     .07       0
#Block Obstruct= 2 ,-1
 8344.83 8524.74   16.78    4365    4440    16.7
Bank Sta=4949.78,5028.41
XS Rating Curve= 0
Exp/Cntr=.3,.1

Type RM Length L Ch R = 1 ,5857.266,1114.29,1136.89,1170.69
XS GIS Cut Line= 6
     3202729.494     13758123.06     3200298.838    13756924.652
      3200177.75      13756873.6     3200108.443    13756838.067
     3199832.475     13756718.78     3198009.368    13754813.061
#Sta/Elev= 30
 2121.14   17.45 2567.13   15.72  2943.1   17.65 4188.11   15.58 4230.64   18.42
 4271.99   19.26 4332.68   18.36  4374.8   15.75 4581.22   17.71 4735.02    14.3
 4826.35   15.73 4961.06   15.15 4974.78   11.44  4991.5    4.67 4992.76     3.1
 4998.36    2.18 5022.35    8.79 5038.94      15 5056.62   16.27 5484.65   14.89
 5621.03   16.54 5946.14   15.11 7350.64   16.62 7416.13   15.79 7457.65    7.43
 7478.41    6.87 7499.17     8.8 7540.68   16.39 7744.14   16.23 7978.44   16.79
#Mann= 4 ,-1 , 0
 2121.14     .07       0 4961.06    .035       0 5038.94     .07       0
 7744.14     .12       0
#Block Obstruct= 2 ,-1
 7349.27 7542.65   16.34    4678    4804      15
Bank Sta=4961.06,5038.94
XS Rating Curve= 0
Exp/Cntr=.3,.1

Type RM Length L Ch R = 1 ,4720.374,30.01,30.01,30.19
XS GIS Cut Line= 6
     3203365.855     13757337.43     3200968.222    13756019.372
     3200679.246    13755857.125     3200379.191    13755684.799
     3199831.902    13755378.879     3198314.009    13754585.119
#Sta/Elev= 30
 1913.32   18.15 2645.43   15.21 3524.26   16.16 4157.13   15.74 4239.63   18.96
 4334.88   14.35 4400.49   16.17 4956.64   13.16 4979.34    6.46 4991.05    6.11
 4991.83    3.53 4993.96    1.92 5016.26    1.97 5029.16    9.91 5189.43   12.54
 5261.23   11.24 5579.26   13.87 5805.95   11.59  5936.7   14.77  6454.5   15.55
 6554.37   14.62 6590.33    6.61 6615.99    5.11 6631.08    9.14 6666.77   16.02
 6734.48   14.43 6947.23   15.31 7200.02   19.94 7463.27   16.15 7666.68    15.8
#Mann= 6 ,-1 , 0
 1913.32     .07       0 3524.26     .12       0 4157.13     .07       0
 4956.64    .035       0 5029.16     .07       0 6631.08     .12       0
#Block Obstruct= 2 ,-1
 6553.12 6660.72   14.59    5620    5960    12.4
Bank Sta=4956.64,5029.16
XS Rating Curve= 0
Exp/Cntr=.5,.3

Type RM Length L Ch R = 1 ,4690.362,40.01,40.01,40.26
XS GIS Cut Line= 6
     3203379.785    13757306.785     3200982.773    13755993.136
     3200694.057    13755831.035     3200393.981    13755658.697
     3199846.194    13755352.498     3198347.982    13754567.323
#Sta/Elev= 30
 1914.63   17.83  2662.1   15.06 3518.91   16.26 4149.16   15.34 4237.24   18.95
 4332.49   14.53 4410.68   16.29 4956.64   13.16 4985.38    6.11 4985.81    4.67
 4985.81    2.38 4993.96    1.92 5024.78    2.37  5025.8    5.78 5029.16    9.91
 5115.73   12.16 5805.13   11.56 5937.86   14.71 6555.59   14.81  6577.9   12.84
 6597.51    6.53  6617.1    4.81  6635.9    5.89 6665.25   14.77 6682.18   16.01
 6964.53   15.52 7089.06   19.33 7205.17   19.76 7402.81   16.39 7644.21   15.77
#Mann= 6 ,-1 , 0
 1914.63     .07       0 3518.91     .12       0 4149.16     .07       0
 4956.64    .035       0 5029.16     .07       0 6555.59     .12       0
#XS Ineff= 2 , 0
       0    4976   10.22    5033       0    9.72
Permanent Ineff=
       F       F
#Block Obstruct= 2 ,-1
 6562.93 6680.01   14.77    5555    5940    12.3
Bank Sta=4956.64,5029.16
XS Rating Curve= 0
Exp/Cntr=.5,.3

Type RM Length L Ch R = 2 ,4669    ,,,
BEGIN DESCRIPTION:
FOREST PARK CEMETARY RD
END DESCRIPTION:
Bridge Culvert--1,0,-1,-1, 0
Deck Dist Width WeirC Skew NumUp NumDn MinLoCord MaxHiCord MaxSubmerge Is_Ogee
10,22,2.6,0, 20, 20, , , .95, 0, 0,0,,
    4171    4232    4289    4352    4498    4570    4656    4807 4860.15 4909.97
 4956.46 5068.53 5114.58    5156    5249    5367    5497    5622    5764    5824
   16.88   18.65   17.47   15.16   15.39   14.66   14.59    13.9   13.59   12.13
    11.4   10.45   11.52    11.9   11.36   12.37   12.61   12.68    12.3   12.03
                                                                                
                                                                                
    4171    4232    4289    4352    4498    4570    4656    4807 4860.15 4909.97
 4956.46 5068.53 5114.58    5156    5249    5367    5497    5622    5764    5824
   16.88   18.65   17.47   15.16   15.39   14.66   14.59    13.9   13.59   12.13
    11.4   10.45   11.52    11.9   11.36   12.37   12.61   12.68    12.3   12.03
                                                                                
                                                                                
Multiple Barrel Culv=2,6.6,12,35,.012,.5,1,8,1,2.72,2.62, 3,Culvert #1  , 0 ,5
  4992.5  4992.5    5005    5005  5017.5  5017.5
Culvert Bottom n=.012
BC Design=,, 0 ,, 0 ,,,,,,
BC HTab HWMax=19.76

Type RM Length L Ch R = 1 ,4650.352,120.04,120.01,120.77
XS GIS Cut Line= 6
     3203404.859    13757278.925     3201002.174    13755958.156
     3200713.805    13755796.249     3200413.701    13755623.895
     3199865.249    13755317.325     3198391.661    13754544.675
#Sta/Elev= 30
 1907.63    16.8  2726.9   14.84 3449.53   16.15 3631.51   18.25 3668.23   15.58
 4134.82   15.04 4253.96   18.58 4332.54   14.78 4421.39   16.41 4956.64   13.16
  4985.7    6.12 4986.04     2.4 4993.96    1.92 5025.04    2.39 5029.16    9.91
 5115.73   12.16 5808.24   11.57 5942.95   14.64 6419.12   15.65 6587.01   14.78
 6620.88     6.6 6637.82    4.68 6660.47    6.51 6688.63   14.76 6714.15   15.33
 6960.35   16.11 7089.08    19.5 7253.44   19.36 7359.32   16.26 7618.38   16.42
#Mann= 6 ,-1 , 0
 1907.63     .07       0 3449.53     .12       0 4134.82     .07       0
 4956.64    .035       0 5029.16     .07       0 6419.12     .12       0
#XS Ineff= 2 , 0
       0    4976   10.22    5033       0    9.72
Permanent Ineff=
       F       F
#Block Obstruct= 2 ,-1
 6583.83 6692.52   14.72    5780    5830    11.9
Bank Sta=4956.64,5029.16
XS Rating Curve= 0
Exp/Cntr=.5,.3

Type RM Length L Ch R = 1 ,4530.347,686.57,690.34,684.14
XS GIS Cut Line= 6
     3203457.792    13757170.273     3201060.377    13755853.214
     3200773.047    13755691.891     3200472.862     13755519.49
     3199922.414    13755211.804     3198519.463     13754476.73
#Sta/Elev= 30
 1920.03   15.56  3213.9      16 3425.21   18.21 3459.41   16.14  3526.4      18
 4113.98   15.29 4228.77   18.74 4331.91   15.54  4657.6   16.74    4954      12
 4991.05    6.11 4993.96    1.92 5016.26    1.97 5020.66    5.82    5051    9.91
    5087   11.38 5469.71   15.24 5726.29   14.84 5815.82   11.77 5989.39   14.86
 6307.94   14.28 6658.63   14.25 6693.83    5.53 6726.37    6.17 6760.24    15.1
 6926.55   15.48 6977.13   19.01 7207.81   18.88 7280.15   15.71 7545.55   16.75
#Mann= 6 ,-1 , 0
 1920.03     .07       0  3213.9     .12       0 4113.98     .07       0
    4954    .035       0    5087     .07       0 6307.94     .12       0
#Block Obstruct= 1 ,-1
 6653.53 6762.97   14.26
Bank Sta=4954,5087
XS Rating Curve= 0
Exp/Cntr=.3,.1

Type RM Length L Ch R = 1 ,3840.003,492.48,585.14,677.52
XS GIS Cut Line= 6
      3201870.41    13755472.187     3201361.903    13755236.455
     3201304.476    13755203.353     3201146.106    13755108.334
     3200896.248    13754974.864     3199266.862    13754078.764
#Sta/Elev= 30
 4138.83   15.51 4275.75   17.66 4339.59   13.62 4479.45   15.82 4518.38   13.52
    4665    14.7 4859.19   13.11 4906.84   11.73 5019.14     1.6  5021.4    2.68
 5022.21    4.71 5048.82    6.79 5190.44   12.72 5320.54   14.27 5374.46   16.13
 5426.13   14.17 5538.33   14.46 5672.58    20.5 5734.14    18.4 5881.85   15.39
 6203.44    13.7 6260.69   10.27 6335.99    9.14 6852.95   15.15 6998.13   14.28
 7036.76    5.32 7049.49    4.11 7066.61    4.64 7083.73    7.53 7093.11   11.02
#Mann= 6 ,-1 , 0
 4138.83     .07       0 4859.19    .035       0 5190.44     .07       0
 5320.54     .12       0 5734.14     .07       0 5881.85     .12       0
#Block Obstruct= 1 ,-1
 5672.96 7309.25   20.49
Bank Sta=4859.19,5190.44
XS Rating Curve= 0
Exp/Cntr=.3,.1

Type RM Length L Ch R = 1 ,3254.865,210.32,515.35,778.31
XS GIS Cut Line= 6
     3201846.836    13755091.649     3201628.545    13754783.888
     3201479.134    13754654.157     3201403.913    13754566.879
     3201289.419    13754433.874     3200315.161    13753522.259
#Sta/Elev= 30
 4367.46   13.96 4482.74   15.08 4549.92   12.15 4631.33   14.43 4688.44   14.57
 4781.51   11.29 4827.34   12.03 4873.58   10.91 4917.05     8.1 4942.39       6
 4953.55    4.29 4954.01    3.03 4956.55    2.34 5044.52    2.02 5047.58     3.5
 5048.05    4.93 5101.35   11.46 5191.93   13.72 5291.53   13.33 5394.24   16.33
 5477.58   14.38    5761   14.55 5911.74    10.8 5999.43   11.58 6095.16   10.48
 6177.05    5.83  6232.6    6.48 6314.83    3.39 6436.85     2.2 6567.62    2.45
#Mann= 4 ,-1 , 0
 4367.46     .07       0 4827.34    .035       0 5101.35     .07       0
 5291.53     .12       0
#Block Obstruct= 1 ,-1
 5397.46 6802.39   16.35
Bank Sta=4827.34,5101.35
XS Rating Curve= 0
Exp/Cntr=.3,.1
